HEC-RAS study PenFrkFshCk.prj: PenFrkFshCk

--- PenFrkFshCk.g01 (geometry) --- (continued)

Type RM Length L Ch R = 1 ,37501   ,281.2,300,317.2
XS GIS Cut Line= 6
1676201.39155951455901.2492565071676280.08201893455838.440983176
1676339.34043059 455784.297390671676401.63361309 455706.06920068
1676448.35267976455647.3980581761676502.85847625455578.948391929
#Sta/Elev= 30
       0     942    12.8  932.65    27.8  924.92    35.6  922.19    48.2  919.57
   111.8  917.85     135  917.68   146.6  918.59   160.6   918.5   165.2  918.19
   179.9  915.35  211.22 913.409   239.9  912.03   249.2  912.54  252.66913.4062
   258.5  917.36   260.9  918.15   291.2  917.62   297.5  918.92   302.9  922.59
   314.9  933.39   325.5   940.8   335.6  949.62   346.5  957.64   360.4  966.38
   372.9  973.43   393.9  983.88   402.3  987.13   427.5  993.85   443.5  996.05
#Mann= 3 ,-1,0
       0      .1       0  211.22    .045       0  252.66      .1       0
Bank Sta=211.22,252.66
XS Rating Curve= 0 ,0
Exp/Cntr(USF)=0,0
Exp/Cntr=0.3,0.1

Type RM Length L Ch R = 1 ,37201   ,301.7,300,299.2
XS GIS Cut Line= 6
  1676215.169091456030.318224087  1676302.661042456029.135483667
1676377.65433034456028.1220342521676477.64527209456026.770987093
1676552.63856043456025.7572095841676640.13051142456024.575125337
#Sta/Elev= 30
       0  946.73     4.2  944.84    16.4  936.57    27.2  930.23      37  925.52
    43.6  923.46    66.6  919.98    79.7  918.82   115.8  917.74   135.5  916.09
   155.2  916.15     165  914.83   174.8  912.22  196.26911.7598   217.9  911.25
  234.71911.7609   243.7  916.16   253.6  919.94   263.4   928.2   283.1  942.57
   306.1  964.64   322.5  985.03     352 1010.94   358.6 1014.93   371.7 1020.95
   394.7 1026.05     398 1027.49   414.4 1037.68   420.8 1042.88     425 1047.26
#Mann= 3 ,-1,0
       0      .1       0  196.26    .045       0  234.71      .1       0
Bank Sta=196.26,234.71
XS Rating Curve= 0 ,0
Exp/Cntr(USF)=0,0
Exp/Cntr=0.3,0.1

Type RM Length L Ch R = 1 ,36901   ,281.7,300,311.3
XS GIS Cut Line= 6
1676216.66121401456328.4629690051676304.50322993456333.385531336
1676379.41515359456329.7490556691676479.29749976456324.900312096
1676554.20909534456321.2638364291676641.60623026 456317.02139084
#Sta/Elev= 30
       0  934.02    12.6  933.82    19.2   933.1    22.4  931.89    35.6  924.12
    42.2  922.12    84.6  921.04   137.4   917.3   157.1  918.94   163.7  916.06
     167   915.1   173.6  914.39  181.37911.3676   186.7  910.32   199.8  909.97
   226.1  910.02   229.4  910.18  234.61911.3668   252.4  916.62   265.5  916.04
     282  916.54   288.5  917.44   298.4   920.3   308.2  925.55   327.9  934.64
   344.4  940.63   348.6  941.85   367.4  945.23   384.5  950.76   425.5  961.74
#Mann= 3 ,-1,0
       0      .1       0  181.37    .045       0  234.61      .1       0
Bank Sta=181.37,234.61
XS Rating Curve= 0 ,0
Exp/Cntr(USF)=0,0
Exp/Cntr=0.3,0.1

Type RM Length L Ch R = 1 ,36601   ,289.3,301.9,310.4
XS GIS Cut Line= 6
1676134.38447568456490.7677625121676208.93353917456536.717145666
1676273.92520709456574.1573595111676361.11728993456623.121828511
1676426.51151609456659.8455083371676502.80467059 456702.68958275
#Sta/Elev= 30
       0  934.71     7.4  934.54    11.2  933.01    23.3  925.75      40  921.93
    57.5  919.71    80.6  918.34   119.6  917.03   133.4  915.75   169.4  915.06
     179  913.69  187.09910.8426   192.4  910.11  232.78910.8422   235.5  912.07
   236.9  913.59   246.8  928.35   251.3  932.86     273  950.41   276.9  954.32
   284.4  963.11   288.2  966.79   314.5  987.05     326  993.69   344.6 1003.08
   363.4 1015.62   382.2 1025.99   397.3 1032.16   408.6 1034.14   425.1 1040.42
#Mann= 4 ,-1,0
       0     .07       0      40      .1       0  187.09    .045       0
  232.78      .1       0
Bank Sta=187.09,232.78
XS Rating Curve= 0 ,0
Exp/Cntr(USF)=0,0
Exp/Cntr=0.3,0.1

Type RM Length L Ch R = 1 ,36299   ,283.7,298.1,309.7
XS GIS Cut Line= 6
1675981.69252384456658.3045009231676039.15271075456725.074708596
1676087.85996242 456782.674330921676147.07605134456863.348054096
1676189.09926125456925.4693209231676238.12606609456997.944241583
#Sta/Elev= 30
       0  933.92     7.6  931.56    16.5   923.9    19.2  922.32    29.5  919.11
    51.1  917.99    61.1  916.23    87.8  914.79    98.6  916.29   124.4  916.47
   133.2  915.65   141.6  913.66   151.9  913.26  180.52909.2122   219.8  908.29
   230.6  908.39  235.05909.2106   250.3  914.36   260.8  916.47   268.8  921.19
   280.7  935.41   304.6  954.53   318.8  969.77   334.1  984.46     344  995.86
   347.1  998.32   369.2  1012.9     392 1025.75   403.8 1030.25   426.1 1037.21
#Mann= 3 ,-1,0
       0      .1       0  180.52    .045       0  235.05      .1       0
Bank Sta=180.52,235.05
XS Rating Curve= 0 ,0
Exp/Cntr(USF)=0,0
Exp/Cntr=0.3,0.1

Type RM Length L Ch R = 1 ,36001   ,278.8,299.3,321.1
XS GIS Cut Line= 6
1675833.03829359456740.4883916681675837.78959642 456829.82876417
1675846.67540543456904.3177884221675860.63896017457003.337931588
1675871.11203635457077.6032029991675883.33051585457164.246074334
#Sta/Elev= 30
       0  927.32    12.4  925.62    28.8  920.61    41.9  917.85    58.3  915.57
    84.6  913.95   107.7  914.03   137.5  915.51     154  912.81   167.2  913.61
   173.8  913.09  188.42 908.872   193.7  907.67   213.6  907.56   235.4   907.7
  239.93908.8699   246.7  918.91     250   922.8   283.2   945.2   290.6  951.56
     308  968.62   334.1  988.08   342.8  993.76   359.4  1002.4   366.1 1006.62
   375.9 1014.18   405.8  1029.7   415.7  1037.4     419 1039.01     427 1040.64
#Mann= 3 ,-1,0
       0      .1       0  188.42    .045       0  239.93      .1       0
Bank Sta=188.42,239.93
XS Rating Curve= 0 ,0
Exp/Cntr(USF)=0,0
Exp/Cntr=0.3,0.1

Type RM Length L Ch R = 1 ,35702   ,252.8,247.7,233.1
XS GIS Cut Line= 6
1675693.54546234456691.4199202511675643.82508934456763.463739425
1675601.41933426456825.3527232561675546.98899692456909.241663083
1675518.07862167 456979.890471921675487.61345951 457064.43295376
#Sta/Elev= 30
       0  939.69     6.8  939.19    14.8  937.59    22.8  934.62    42.7  929.18
    62.6  920.68    81.2  916.57   106.5  913.88   154.2  913.14     166  911.47
   173.9  911.51  184.06908.5495   238.7  907.47   251.6  907.71  255.31908.5506
   267.2  912.23   282.2  912.63   291.2  913.75   316.9  925.56   331.1   929.5
   341.6  933.08   349.2  934.75   355.6   937.3   369.5  946.52   383.5  954.15
     387  957.02   397.4  967.82   404.4  973.95   411.4  979.28   428.8  995.96
#Mann= 3 ,-1,0
       0      .1       0  184.06    .045       0  255.31      .1       0
Bank Sta=184.06,255.31
XS Rating Curve= 0 ,0
Exp/Cntr(USF)=0,0
Exp/Cntr=0.3,0.1

Type RM Length L Ch R = 1 ,35454   ,340.9,348.4,356.7
XS GIS Cut Line= 2
  1675449.123617456539.3432250471675272.88021946456987.245742219
#Sta/Elev= 30
       0  958.89     8.3  955.82    17.9  953.35    56.7  947.81    91.9  940.27
   102.5   937.2   127.2  936.32   130.7  934.73   148.3  920.62   162.4  914.11
   165.9  913.38   197.7  911.91   208.3  909.95   213.9  908.15   218.3   907.3
   229.4  907.12   296.4  907.44   301.4  908.14     307  910.01   319.5  911.76
   342.2  911.37   349.3  912.12   366.9  917.71   377.7  920.31   410.6  925.48
   423.3  931.16   437.4  934.72   451.5  944.38   472.7  955.71   481.3  962.49
#Mann= 3 ,-1,0
       0      .1       0   213.9    .045       0   301.4      .1       0
Bank Sta=213.9,301.4
XS Rating Curve= 0 ,0
Exp/Cntr(USF)=0,0
Exp/Cntr=0.3,0.1

Type RM Length L Ch R = 1 ,35106   ,300.3,300,299.2
XS GIS Cut Line= 6
1675190.70919767456384.8650871661675150.23519726456462.441375583
1675115.54268134456528.9353370821675069.28621218456617.593952417
1675035.21672651456684.4127164191674953.00835852456860.119932069
#Sta/Elev= 30
       0  999.81    52.4  972.97    70.9  962.14   108.5   945.4   126.4  935.13
   130.1  934.28     145  934.36     162  920.91   166.8  918.63   174.5  916.91
   178.2  914.05   181.9  909.66   185.6  906.96  192.74905.0956   208.2  904.41
  244.68905.0966   259.6  909.07   281.2   909.2   314.9  910.88   351.5  909.57
   362.3  908.44   384.1   909.6   416.7  909.17   427.5  908.17   452.9  909.37
   463.7  911.99     500  925.93   507.2   930.4   518.1  940.09   531.5  950.54
#Mann= 3 ,-1,0
       0      .1       0  192.74    .045       0  244.68      .1       0
Bank Sta=192.74,244.68
XS Rating Curve= 0 ,0
Exp/Cntr(USF)=0,0
Exp/Cntr=0.3,0.1

Type RM Length L Ch R = 1 ,34806   ,305.6,300,292.2
XS GIS Cut Line= 6
1674914.44006518456260.5579210821674875.30858175456338.820231751
1674841.76731026456405.9021185931674797.04561493456495.344525009
1674763.50434342456562.4264118371674649.22525944456780.551562052
#Sta/Elev= 30
       0 1001.17    25.2  990.43    58.9  973.86    69.2  966.74    77.2  960.01
    91.9  951.47   101.2  942.75   110.2  937.19   145.2  935.88   161.6  931.78
   172.6  921.64   191.4  906.73  195.39904.5047   201.9  903.19   229.2  903.16
  242.19904.5038   262.5  907.63   275.3  907.25   286.3  908.39   379.5  909.54
   411.7   907.2   430.2  908.12   474.7   907.6   496.1  909.16   510.7  913.99
   526.5  916.97   533.9  920.27   544.8  928.15   563.6  946.08   583.7   959.3
#Mann= 3 ,-1,0
       0      .1       0  195.39    .045       0  242.19      .1       0
Bank Sta=195.39,242.19
XS Rating Curve= 0 ,0
Exp/Cntr(USF)=0,0
Exp/Cntr=0.3,0.1

Type RM Length L Ch R = 1 ,34506   ,293.1,300,307.6
XS GIS Cut Line= 6
1674573.96699284456155.9186946751674557.01099001456241.760058418
1674542.47689834456315.3379952611674523.09832817 456413.44245784
1674508.56456459456487.020722762 1674467.0691466456731.422341469
#Sta/Elev= 30
       0  1011.3    16.5 1005.17    53.3  980.82      57   977.1    63.3  965.64
      70  956.59    90.1  937.11    93.4  934.89   103.5   935.4   120.2  932.95
   130.2     933   143.6  929.84   146.9  928.14     167  909.54   170.3  907.59
   177.1  906.61  185.33 903.582   193.7  903.06  238.87903.5819     254  906.14
   284.1  907.79   370.8  908.91   400.8  906.46   410.8  907.61   450.7  907.05
   510.6  908.58   520.6  913.42   547.2  939.69   580.5  964.67   585.4  969.54
#Mann= 3 ,-1,0
       0      .1       0  185.33    .045       0  238.87      .1       0
Bank Sta=185.33,238.87
XS Rating Curve= 0 ,0
Exp/Cntr(USF)=0,0
Exp/Cntr=0.3,0.1

Type RM Length L Ch R = 1 ,34206   ,385.6,371.3,355
XS GIS Cut Line= 6
1674351.62787059456067.4543046651674311.49671726456145.208742335
1674277.09849209456211.8552625921674231.23441058456300.717289582
1674139.93505875456539.726301549 1674225.6922334456762.771892851
#Sta/Elev= 30
       0 1037.66    18.1 1031.36    47.7 1011.02    62.4 1002.83    73.5  989.58
    80.9  977.12    91.9  955.39   114.1  936.48   117.8  934.99     151  933.04
   165.8  924.97   176.9  915.82   187.9  904.19  193.74901.8269   224.9   900.8
  242.48 901.828   265.3  905.99   286.4  904.65   297.6  906.06   437.5  908.44
   539.3  912.36   588.5  911.73   606.1  913.31   614.3  916.89   634.2  935.69
   648.2  945.01     663  952.14   680.3  957.03     698   966.8   757.3  990.48
#Mann= 5 ,-1,0
       0      .1       0  193.74    .045       0  242.48      .1       0
   492.5     .05       0  558.35      .1       0
Bank Sta=193.74,242.48
XS Rating Curve= 0 ,0
Exp/Cntr(USF)=0,0
Exp/Cntr=0.3,0.1

Type RM Length L Ch R = 1 ,33835   ,230.5,228.7,228.6
XS GIS Cut Line= 6
1673840.14925886456007.5434616731673882.90540694456164.317426331
1673902.02643169456262.7552215831673908.92438377456338.613009505
1673943.45247614456529.4387611971673887.97388293456736.870517765
#Sta/Elev= 30
       0 1032.83    14.2 1023.38    30.4 1004.32    41.4   995.3    65.2  970.47
    75.4  955.35    92.4  938.69    99.2  935.71   119.6  935.04   153.6  920.61
   167.1  917.09     178  910.87  190.37 900.639   220.6  899.66  233.31900.6401
     264  905.83   393.1  903.06   406.5  906.35   509.2  908.35     540  911.53
   570.5  920.04   584.1  925.42   592.8  926.77   607.9  936.98   624.9  941.47
   635.7  949.31     669  964.75   696.2  983.66   713.2  989.36   747.6 1008.11
#Mann= 7 ,-1,0
       0      .1       0  190.37    .045       0  233.31      .1       0
  302.78     .05       0  518.95      .1       0  528.95     .05       0
  542.87      .1       0
Bank Sta=190.37,233.31
XS Rating Curve= 0 ,0
Exp/Cntr(USF)=0,0
Exp/Cntr=0.3,0.1

Type RM Length L Ch R = 1 ,33606   ,305.3,300,293.5
XS GIS Cut Line= 6
1673618.82224959456076.4769244191673660.78870109456233.464143261
1673686.61476493456330.0718896691673705.98382068456402.527781501
1673720.71307036456453.9338778811673787.09750099456687.147377377
#Sta/Elev= 30
       0 1025.71    20.9 1002.17    41.3   985.3    54.9  966.43    61.6  953.29
      65  949.12    75.2  940.02    82.6  935.84    93.3   935.4   105.8  930.67
     116  930.65   138.8  916.91   160.1  909.06   173.7  905.73  184.59 899.826
   190.7  899.01  244.22 899.824   251.8  905.28   329.1  901.89   350.4  903.78
   449.3  906.52   473.2  909.24   500.5  918.18   517.5  920.39   522.1  921.93
   565.3  946.01   599.4  959.12   616.5   972.9   626.7  975.35   633.5  979.87
#Mann= 5 ,-1,0
       0      .1       0  184.59    .045       0  244.22      .1       0
   272.5     .05       0  490.97      .1       0
Bank Sta=184.59,244.22
XS Rating Curve= 0 ,0
Exp/Cntr(USF)=0,0
Exp/Cntr=0.3,0.1

Type RM Length L Ch R = 1 ,33306   ,298.1,300,302.4
XS GIS Cut Line= 6
  1673301.718225456206.4202340841673341.04951118456284.582151249
1673374.76237026456351.578080252 1673419.7124116456440.905985594
 1673453.4249426456507.9019145821673555.04808558456714.422133399
#Sta/Elev= 30
       0 1036.63    16.7 1032.61    31.4 1026.35    68.1  997.14    71.8  991.53
    79.1  975.24    90.1  956.02   108.5  940.72   112.2  938.24   119.5  935.77
     134  933.51   145.2  933.79   152.6  930.87   178.3  910.46   187.8  900.83
     192898.4669   207.7  897.66  242.54898.4658   259.1  902.99   299.5  901.36
   405.5  906.33   422.6  908.27   431.3  909.98   442.4  914.06     457  915.74
   475.2  924.58     501  944.33   523.1  955.72   548.3   974.3   567.7  986.18
#Mann= 5 ,-1,0
       0      .1       0     192    .045       0  242.54      .1       0
   312.5     .05       0   417.5      .1       0
Bank Sta=192,242.54
XS Rating Curve= 0 ,0
Exp/Cntr(USF)=0,0
Exp/Cntr=0.3,0.1

Type RM Length L Ch R = 1 ,33006   ,299.2,300,300.6
XS GIS Cut Line= 6
1673044.08521008456320.2375917581673076.62910825456401.460198343
1673104.52406558456471.079809755 1673141.7169046456563.905739591
1673169.61186193456633.5253510031673255.00950649456844.994209386
#Sta/Elev= 30
       0  939.71      56  936.95    70.2  937.23    87.8  934.71   127.9  934.11
   133.8  933.29     138     932   144.4  928.16   157.4  915.63   172.7  905.79
   179.7  899.52  182.75897.8958   186.8  897.02   216.2  896.59  232.77897.8957
   243.4  901.73   268.1  902.98     314  902.87   335.2   901.4     354  903.11
   395.4  904.63   409.5  906.47   423.7  911.05   434.3  912.55   444.9  918.46
   473.5  931.07   496.1   944.9   515.7  954.19   540.5  970.92   565.6  984.66
#Mann= 3 ,-1,0
       0      .1       0  182.75    .045       0  232.77      .1       0
Bank Sta=182.75,232.77
XS Rating Curve= 0 ,0
Exp/Cntr(USF)=0,0
Exp/Cntr=0.3,0.1

Type RM Length L Ch R = 1 ,32706   ,419.6,422.8,420.1
XS GIS Cut Line= 6
  1672775.900379456443.650074586 1672806.7864721456525.517364919
1672833.26017243456595.6897967611672868.55865826456689.252601758
1672895.03235859456759.4247055051672971.22138166456963.987759306
#Sta/Elev= 30
       0  978.31     7.8  970.73    11.3  968.94    21.9  966.92    30.1  963.26
    75.9  938.05    91.2  934.42     113  934.23   116.5  933.15   144.6  912.22
   169.1  902.51   176.2  898.22  181.92897.0203   214.7  896.39  235.98897.0212
   246.3  901.37   256.8  902.13   281.4  902.19   298.9  900.72   316.4  902.01
   333.9  901.06   389.2  904.31   427.5  909.92   449.5  916.37     460  921.25
     467  926.16   484.5  941.43     502  953.97     516  966.61   555.8  996.02
#Mann= 5 ,-1,0
       0      .1       0  181.92    .045       0  235.98      .1       0
   272.5     .05       0   367.5      .1       0
Bank Sta=181.92,235.98
XS Rating Curve= 0 ,0
Exp/Cntr(USF)=0,0
Exp/Cntr=0.3,0.1

Type RM Length L Ch R = 1 ,32283   ,375.3,384.2,383.9
XS GIS Cut Line= 2
1672398.45392577456608.5823585021672601.57064812457098.762547961
#Sta/Elev= 30
       0  964.12    24.1  961.08    28.3  959.81    35.4   956.1    54.2   942.5
    63.8  937.33    74.5  933.56     107  932.14     112  928.11   120.6  916.65
   124.5  912.43   134.8  905.11   152.6  898.67   167.2  898.27  177.65895.9301
   223.6   894.9   237.5  895.75   248.5  894.76  263.38895.9318   276.9  900.33
   307.8  898.87   326.6  898.99   337.2  904.07   340.8  904.77   422.5     910
   432.6  914.47   468.5  941.96     494  953.61   518.4  967.14   530.6  972.25
#Mann= 4 ,-1,0
       0      .1       0     160     .06       0  177.65    .045       0
  263.38      .1       0
Bank Sta=177.65,263.38
XS Rating Curve= 0 ,0
Exp/Cntr(USF)=0,0
Exp/Cntr=0.3,0.1

Type RM Length L Ch R = 1 ,31899   ,391.2,393,394.7
XS GIS Cut Line= 6
1672045.09365965456706.6677733371672075.12312715456788.853632585
1672100.86290507456859.2983735961672135.18239024456953.224694923
1672160.92184007457023.6697640131672219.26531073457175.697640329
#Sta/Elev= 30
       0  945.13    66.6  940.08    72.7  938.43    80.6  933.98    87.5  933.09
    94.5  930.64     119  929.52   122.5  928.11     126  924.99   146.9   902.6
   150.4   900.8   160.9  898.93  169.75895.4755   178.4   894.2   220.3  894.77
  224.52895.4744   230.8  898.79   234.3  899.01   258.7  899.32   286.7   898.1
   304.1  899.95   363.7  899.81   384.7  901.36   394.6  905.92   405.8  907.97
   444.5  928.74   475.9  946.88   483.1  954.59   488.1  958.83   500.3   966.8
#Mann= 3 ,-1,0
       0      .1       0  169.75    .045       0  224.52      .1       0
Bank Sta=169.75,224.52
XS Rating Curve= 0 ,0
Exp/Cntr(USF)=0,0
Exp/Cntr=0.3,0.1

Type RM Length L Ch R = 1 ,31506   ,301,300,299.3
XS GIS Cut Line= 6
1671677.78577735456802.3668768411671702.28572834456886.366708845
1671723.28568634456958.3668929191671751.28563035457054.367029011
1671772.28558834457126.3668850061671817.54938225457285.871600327
#Sta/Elev= 30
       0  963.62    20.2  961.11    44.1  950.67    71.4   943.5    95.3  929.64
   115.8  927.95   132.8  928.47   146.6  927.26   156.9  921.13   173.9  904.87
   180.4  896.83  186.53894.0853   225.2  893.41  235.11894.0849     249   895.3
   259.8   898.9   320.7  898.22   341.8   895.8   368.7  895.16   384.3  898.75
   406.2  900.56     413  903.61   419.8  908.22   440.3  925.24   443.7   926.8
   453.9   928.4   460.8  932.28     471  941.12   484.6   955.1   503.3  967.84
#Mann= 3 ,-1,0
       0      .1       0  186.53    .045       0  235.11      .1       0
Bank Sta=186.53,235.11
XS Rating Curve= 0 ,0
Exp/Cntr(USF)=0,0
Exp/Cntr=0.3,0.1

Type RM Length L Ch R = 1 ,31206   ,304.2,298.7,292.5
XS GIS Cut Line= 6
1671388.61345543456903.0422004161671415.74069776456986.231010422
 1671438.9919636457057.5356578381671469.99387009457152.608630419
1671493.24513592457223.9136059281671558.12481992 457418.47211881
#Sta/Elev= 30
       0  943.49    28.3   936.4    92.8  925.33   103.2  924.48   128.4  919.06
   159.5  909.83   169.8  903.01   180.2  899.23   187.1  894.79  192.17892.8735
   197.4  891.93   228.5  891.81  238.33892.8744   252.6  895.34   280.1  894.22
   304.4  898.23   383.9   896.5   394.3  897.34   418.5  897.49   432.3  899.12
   440.6  903.08   463.4  919.48   470.3  923.76   473.8  925.45   482.6  927.63
   490.4   931.3   502.8  941.29   511.8   947.6   525.7   955.7   542.6  964.39
#Mann= 3 ,-1,0
       0      .1       0  192.17    .045       0  238.33      .1       0
Bank Sta=192.17,238.33
XS Rating Curve= 0 ,0
Exp/Cntr(USF)=0,0
Exp/Cntr=0.3,0.1

Type RM Length L Ch R = 1 ,30907   ,316.2,301.3,281.5
XS GIS Cut Line= 6
1671068.76271717457040.0435668381671114.11367634457114.873469666
1671152.98597392457179.0134332631671207.08101009457263.160902753
1671255.57402334457321.4701693361671420.52565082457503.220467563
#Sta/Elev= 30
       0  972.55    17.1  965.65    43.9  951.44    59.3   940.1    72.6  937.69
    89.3   931.2   101.2  924.24   108.4  922.77   132.5  922.03   155.2  915.41
   164.1  909.85   177.6  898.62  189.74892.0908   204.4  891.28   229.2  891.28
  235.37892.0913   248.8  895.22   281.5  899.65   360.8  898.12     399  898.84
   431.1  898.11   437.5  897.66   449.1  894.74   469.8  896.06   495.5  895.97
   507.1   899.5   523.8  909.44   539.7  920.16   553.6  922.57   583.8  942.27
#Mann= 5 ,-1,0
       0      .1       0  189.74    .045       0  235.37      .1       0
   262.5     .05       0  508.37      .1       0
Bank Sta=189.74,235.37
XS Rating Curve= 0 ,0
Exp/Cntr(USF)=0,0
Exp/Cntr=0.3,0.1

Type RM Length L Ch R = 1 ,30606   ,315,300,277.8
XS GIS Cut Line= 6
1670827.04436859457421.9151784181670911.80863476457443.623140261
1670984.46400125457462.2300584171671081.33749518457487.039063916
1671155.16674384457501.0626579231671374.60752973457539.267886833
#Sta/Elev= 30
       0 1015.33    12.2 1009.05    35.9 1005.61    49.5 1000.35    59.6  994.64
    73.2  984.21    79.9  970.57    86.7  960.72    93.5  948.55   120.6  925.07
   128.5  920.35   140.9  916.86   161.2  916.34   164.6   914.1   171.4  905.81
   174.8  903.82   181.5  902.25   188.3  894.66  194.27891.0876   225.6  890.09
  240.79891.0855   276.2   898.3   372.9  897.35   396.2  894.66   426.2  894.34
   483.8  899.72   499.5  904.39   522.8  918.92   536.1  921.98   560.4  934.11
#Mann= 5 ,-1,0
       0      .1       0  194.27    .045       0  240.79      .1       0
   282.5     .05       0  487.65      .1       0
Bank Sta=194.27,240.79
XS Rating Curve= 0 ,0
Exp/Cntr(USF)=0,0
Exp/Cntr=0.3,0.1

Type RM Length L Ch R = 1 ,30306   ,302.7,300,297.2
XS GIS Cut Line= 6
1670933.15734534 457861.418236421671007.98659201457816.065964922
1671072.12622751 457777.193011181671157.64606959457725.362734258
1671221.78570509457686.4901085941671385.33384582 457663.78995825
#Sta/Elev= 30
       0  961.17    31.5  934.01      41  923.72      47  919.63    55.3   915.8
    73.9  910.99    85.4   910.4    93.1  912.08   100.7   916.4   108.4  918.49
   116.1  919.18   129.4  918.47   136.6  916.06     166  900.71   177.5  892.95
   188.9889.5217   215.4  888.85  235.71889.5232   246.4  892.46   258.4   892.4
   323.3  899.09   341.8   902.2   361.6  906.93   371.6  907.93   384.8     914
   398.2  918.66   431.2  926.86   444.4  933.16   457.7  937.95   502.6  957.38
#Mann= 4 ,-1,0
       0      .1       0      20     .06       0   188.9    .045       0
  235.71      .1       0
Bank Sta=188.9,235.71
XS Rating Curve= 0 ,0
Exp/Cntr(USF)=0,0
Exp/Cntr=0.3,0.1

Type RM Length L Ch R = 1 ,30006   ,311.6,300,286.8
XS GIS Cut Line= 6
1671078.39754042458153.7021006791671146.50895275 458098.77406092
1671204.88974151458051.6924621761671282.73144934457988.917653337
1671341.11256617457941.8363826721671406.68494159457882.902445421
#Sta/Elev= 30
       0  995.33     5.2  992.77      14  986.82    26.1  974.34      49  959.44
    65.3  946.32    80.1  937.46    83.6  934.12    88.8  927.42      94  921.96
   101.1  916.68     119  907.43   141.1  904.75   156.8  904.88     162  904.01
   172.8  898.58   181.2  891.98  189.37887.8735   193.8  887.19   212.3  886.99
   228.6  887.04  233.52887.8755   250.8  892.61   261.3  896.69   270.6  899.15
   286.9  900.86   329.2  902.52   359.2  905.09   381.2  908.31   425.7  916.76
#Mann= 5 ,-1,0
       0      .1       0   137.5     .06       0  189.37    .045       0
  233.52     .06       0   252.5      .1       0
Bank Sta=189.37,233.52
XS Rating Curve= 0 ,0
Exp/Cntr(USF)=0,0
Exp/Cntr=0.3,0.1

Type RM Length L Ch R = 1 ,29706   ,224.4,224.5,220.8
XS GIS Cut Line= 6
1671434.36926943 458356.290606261671463.89709751458273.923645005
1671489.20675817458203.3230644171671522.95275368458109.189066336
1671547.15775776458038.1928172561671572.61275934457954.365229011
#Sta/Elev= 30
       0 1006.27      16  997.94      27  990.79    30.5  987.78    37.4  979.63
    40.9  976.29    82.7   941.6    89.7  931.92    93.2  927.95   100.2  922.85
   131.4  906.04   139.1  903.05   157.1  900.57   166.4  899.99   176.9  900.39
   183.8  899.05   187.3  896.73   194.3  889.25  197.83 887.449   204.7  886.25
   239.6  886.19  251.31887.4471   267.4  891.87   295.2  892.78   312.5  898.82
   350.4  901.47   366.2  903.55   374.5  905.36   405.3  916.68   425.1  921.04
#Mann= 4 ,-1,0
       0      .1       0      60     .06       0  197.83    .045       0
  251.31      .1       0
Bank Sta=197.83,251.31
XS Rating Curve= 0 ,0
Exp/Cntr(USF)=0,0
Exp/Cntr=0.3,0.1

Type RM Length L Ch R = 1 ,29481   ,374.4,375.5,376.2
XS GIS Cut Line= 3
1671667.83592007458410.8227352631671761.43875131458063.667300151
1671820.33442462457965.910161568
#Sta/Elev= 30
       0  977.41    14.8  969.19    28.4  958.86    48.8  948.14    54.6  944.54
    63.4  936.34    82.8  922.36    92.9  913.99   100.9   909.2   114.3  903.66
   120.2  902.04   154.1  897.79   177.9  898.74   181.2  898.07   188.1  894.01
  195.14  887.81   198.3  886.56   201.7  886.35   245.9  886.09   258.8  887.81
   279.9  890.86   290.1  890.16   334.2  892.45   339.1  894.44   355.1  906.63
   361.7  910.06   396.2  916.76   415.4   921.2   449.8  930.12   473.7  937.48
#Mann= 5 ,-1,0
       0      .1       0     140     .06       0  195.14    .045       0
   258.8     .06       0     260      .1       0
Bank Sta=195.14,258.8
XS Rating Curve= 0 ,0
Exp/Cntr(USF)=0,0
Exp/Cntr=0.3,0.1

Type RM Length L Ch R = 1 ,29106   ,298.5,300,302.1
XS GIS Cut Line= 6
1671978.56558268 458453.676743911672034.40087776458320.659772009
1672064.46216933458251.9479671721672104.54411018458160.332008675
1672134.60540175458091.620531917  1672169.677182458011.456650257
#Sta/Elev= 30
       0  922.75    26.4   901.6      30  899.49    33.5  898.71    51.3  898.63
    65.6  896.06    92.8  895.92   101.1  892.74   111.8  890.08   172.5     889
   229.8  889.33  250.99885.3207   257.6  884.29   276.3  883.91     290  884.08
  295.98885.3205   301.4  887.79   312.4  897.78   315.7  903.16   319.8  912.27
   322.3  916.66   326.5  921.02   329.2  922.69   337.2   925.8   378.4  937.81
   387.4  942.81   398.1  950.51   412.4  957.39   451.6  981.06   481.8  992.69
#Mann= 3 ,-1,0
       0      .1       0  250.99    .045       0  295.98      .1       0
Bank Sta=250.99,295.98
XS Rating Curve= 0 ,0
Exp/Cntr(USF)=0,0
Exp/Cntr=0.3,0.1

Type RM Length L Ch R = 1 ,28806   ,285.9,303.6,323.5
XS GIS Cut Line= 6
1672214.85108368458601.3829074871672294.47778542458447.159847096
1672330.09746484458381.1583386661672377.59080817458293.156218082
1672413.21081567458227.1543815881672454.76749109458150.152567089
#Sta/Elev= 30
       0  931.99       9  928.71    12.7  926.24    25.7  910.66    34.9  902.04
      40  899.35    49.7  897.53      57   895.1    80.5   894.2   101.3  890.43
   130.9  887.97   257.2  888.81  280.88 884.338   294.5  883.81  323.44 884.338
   328.1   886.1   331.8  888.82   335.5  892.49   342.5  902.62   347.3  906.88
   371.6  922.64   396.9  938.11   402.6  942.86   413.8  953.74   429.7  964.84
   447.4  979.73   474.1  997.01     495 1009.64   504.7 1015.17   511.1 1017.77
#Mann= 5 ,-1,0
       0      .1       0      30     .06       0     160      .1       0
  280.88    .045       0  323.44      .1       0
Bank Sta=280.88,323.44
XS Rating Curve= 0 ,0
Exp/Cntr(USF)=0,0
Exp/Cntr=0.3,0.1

Type RM Length L Ch R = 1 ,28502   ,285.5,296.4,306.1
XS GIS Cut Line= 6
1672289.62074818458659.4768894941672454.19957884458581.049999252
1672524.68008092458552.3745316711672620.80620101458523.906740844
1672694.04916476458507.7683216781672779.49978125 458488.94060342
#Sta/Elev= 30
       0   925.5     6.6  923.19    13.8  917.52    19.6  911.89    28.4  900.34
      32  897.05    39.3  894.63    54.6  895.03    77.5     898    82.9  896.26
    93.8  890.09     123  885.62   133.8  885.31     181  888.01   224.8   887.6
   248.3  888.53  285.43882.6398   322.1  881.57  335.77 882.641   347.3  887.17
   364.9  899.37   388.4   911.9   419.1  934.83   438.8  945.92   448.9  955.71
   469.1  971.49   492.6  992.26   502.6 1006.72   512.7 1016.72   521.2 1022.54
#Mann= 3 ,-1,0
       0      .1       0  285.43    .045       0  335.77      .1       0
Bank Sta=285.43,335.77
XS Rating Curve= 0 ,0
Exp/Cntr(USF)=0,0
Exp/Cntr=0.3,0.1

Type RM Length L Ch R = 1 ,28206   ,290,300,309.7
XS GIS Cut Line= 6
 1672388.9031215458822.6266158371672476.59848417458824.657123595
1672551.64918709 458827.638744921672651.20935543458837.008804917
1672725.87915359458844.0366780011672812.99446492458852.235808596
#Sta/Elev= 30
       0  898.28     8.4  894.99    21.5  893.47      28  893.62    41.8  897.17
    44.5  896.67    57.6  889.17    64.1  887.92   103.5   884.9   156.1  885.82
   165.9  884.98  177.33882.0438   198.9  881.02   231.8  881.31  236.79882.0436
   241.7  883.41   251.6  889.88   257.8   892.5     278  899.53   291.2  902.52
   296.9  904.88   310.9  913.86   333.1  926.21   347.2  931.96   370.2  948.61
   380.1  954.11   393.3  956.83   396.6  958.48   415.1  973.37   425.3  977.84
#Mann= 5 ,-1,0
       0      .1       0      30     .06       0      60      .1       0
  177.33    .045       0  236.79      .1       0
Bank Sta=177.33,236.79
XS Rating Curve= 0 ,0
Exp/Cntr(USF)=0,0
Exp/Cntr=0.3,0.1

Type RM Length L Ch R = 1 ,27906   ,296,300,304
XS GIS Cut Line= 6
1672331.36058567459019.7987936741672409.09796301459059.962755337
1672475.73004758459094.3888675871672564.57271767459140.291006759
1672631.24974968459174.6298488381672710.48220275459211.900443584
#Sta/Elev= 30
       0  908.46    15.1  901.13    26.2  894.36    29.9  892.77    74.2  891.85
    92.8  892.91   107.4  892.66   114.8  891.45   122.2  887.54   129.3  885.75
   151.7  883.46   166.5  883.97   181.3  883.36  194.14880.9282   202.3  880.26
  240.59880.9299   248.6  884.57   263.2   887.6   280.3  898.14   306.8  909.11
   314.2  912.83   326.5  921.23   332.6  924.56   347.2  929.12   361.7  935.51
   368.3  940.92   376.2  946.31   391.3   954.8   408.8   968.4   425.1  977.76
#Mann= 4 ,-1,0
       0     .06       0   192.5      .1       0  194.14    .045       0
  240.59      .1       0
Bank Sta=194.14,240.59
XS Rating Curve= 0 ,0
Exp/Cntr(USF)=0,0
Exp/Cntr=0.3,0.1

Type RM Length L Ch R = 1 ,27606   ,295,300,305.4
XS GIS Cut Line= 6
1672200.61379993459245.4568069281672270.17205976459298.540690258
1672329.79333159459344.0412554291672409.28857942459404.708456919
1672468.91017935459450.2086940111672539.73451276459501.633459926
#Sta/Elev= 30
       0  899.14    19.1  894.65    53.4  890.89    86.4  890.24   119.4  892.58
   140.1  892.01   156.6  888.45     169  883.56   180.6  882.85  189.85879.4313
   201.4  878.27  235.11879.4318   241.5   881.8     250   888.4   266.3  891.93
   271.7  894.18   282.5  904.66   293.3  913.69     300   918.7   311.7  925.37
   320.3   931.2   323.4  934.77   329.9  943.93     334  947.73   346.9  956.41
   353.3  962.55   381.2  985.13   391.5  994.34   414.7  1008.2     425 1011.56
#Mann= 4 ,-1,0
       0     .06       0  189.85    .045       0  235.11     .06       0
   292.5      .1       0
#XS Ineff= 2 , 0
           119.6  917.87
Permanent Ineff=
       F       F
Bank Sta=189.85,235.11
XS Rating Curve= 0 ,0
Exp/Cntr(USF)=0,0
Exp/Cntr=0.3,0.1

Type RM Length L Ch R = 1 ,27306   ,291.9,301.4,308.9
XS GIS Cut Line= 6
1672056.27813059459450.8297557531672113.08904059 459517.40016067
1672160.66309242459575.3806877581672224.09505217 459652.68794784
1672271.66877593459710.6681468341672327.17161767459778.312040418
#Sta/Elev= 30
       0  894.14      20  893.12      89  893.19   103.7  890.35   117.7  889.49
     134  885.83   152.6  884.31   173.9  884.55   186.6   879.9  191.72 878.679
   214.8  877.43  236.89 878.679   241.8  879.94   245.9  883.81   250.6  890.12
   254.5  892.24     263  888.84   267.2  888.38   283.2  891.99   292.7  892.94
   311.2  897.45   320.5  898.88   328.6  898.95   343.9   903.3   353.2  907.66
   369.5  917.54   388.1  926.23   406.2  933.14     420  936.33     425   938.2
#Mann= 6 ,-1,0
       0     .06       0      50     .07       0  162.52     .06       0
  182.52      .1       0  191.72    .045       0  236.89      .1       0
Bank Sta=191.72,236.89
XS Rating Curve= 0 ,0
Exp/Cntr(USF)=0,0
Exp/Cntr=0.3,0.1

Type RM Length L Ch R = 1 ,27004   ,269.2,289,296.2
XS GIS Cut Line= 6
1671917.58877543459535.6422501651671917.25872359459635.141395003
1671918.94080684459718.8059258461671948.35774276459814.757833675
1671968.34162667459887.0398413391671988.25464459459972.242098749
#Sta/Elev= 30
       0  893.76    41.9  892.78    68.2  890.62     101  884.21   183.2  883.68
  206.83 876.993   241.4  876.23  248.88876.9917   255.1  879.37     262  884.63
   268.8  892.89   275.7  905.01   279.1  909.84   282.5  913.07   289.4   918.1
   309.8  930.67   313.2  933.87     320  942.26   323.4  944.53   338.3  952.49
   347.2  959.26   358.5  965.92   373.3  972.59   384.4  979.04   387.8  980.25
   401.3  982.15   404.6  983.83   415.4  992.77   427.9 1000.78     446 1008.11
#Mann= 5 ,-1,0
       0     .07       0    99.5     .06       0  193.18      .1       0
  206.83    .045       0  248.88      .1       0
Bank Sta=206.83,248.88
XS Rating Curve= 0 ,0
Exp/Cntr(USF)=0,0
Exp/Cntr=0.3,0.1

Type RM Length L Ch R = 1 ,26715   ,314.6,309.5,303.4
XS GIS Cut Line= 6
1671719.12697658459472.560969966 1671703.5082414459560.056201803
1671689.49448991459634.8211441371671660.39776333459730.672330382
1671634.46999366459801.0478457981671604.22071033459883.152996543
#Sta/Elev= 30
       0   915.3    43.4  912.46    61.7  906.23    73.4  904.79      80  901.68
    93.4  891.69   110.1  890.39   116.7  887.35   123.4  882.46   130.1  879.98
   140.1  880.54   156.8  889.82   170.3  892.26   180.6  892.21   190.9  884.39
   198.7  876.37   201.1     875     208  874.51   228.6  874.71   234.6 876.416
   252.6  881.22   276.8  889.69   297.8  894.72   330.9  898.69   360.7  903.96
   374.7  907.71   385.2  912.19   402.4  921.76   413.2  922.36   427.6   929.7
#Mann= 4 ,-1,0
       0     .06       0   198.7    .045       0   234.6     .06       0
  390.12      .1       0
#XS Ineff= 2 , 0
          173.65  897.91
Permanent Ineff=
       F       F
Bank Sta=198.7,234.6
XS Rating Curve= 0 ,0
Exp/Cntr(USF)=0,0
Exp/Cntr=0.3,0.1

Type RM Length L Ch R = 1 ,26406   ,305.5,300,293
XS GIS Cut Line= 6
 1671383.7381371459402.5631200081671380.37528293459489.998312593
1671377.49274276459564.9430445881671373.64957459459664.869025841
1671372.39990517 459739.876421751671371.92484051 459827.42283459
#Sta/Elev= 30
       0  952.72    27.4  939.16    50.4  924.33      57  920.98    73.4  917.04
   106.2  904.28   125.9  898.47   132.5  895.65     139   891.8   142.3  891.03
   165.3  890.61   171.7  889.07   175.2  886.81   181.7     880     185  877.61
  191.35875.0225   211.3  874.11  237.55875.0216   263.8  882.65   276.9  883.57
   286.8  880.84   293.9  880.76   310.5  883.28   322.9  887.36   329.4  890.67
   332.7  891.55   365.5  893.59   383.7   895.6   398.3  897.94   425.1   904.8
#Mann= 5 ,-1,0
       0      .1       0   117.5     .06       0  191.35    .045       0
  237.55     .06       0  417.52      .1       0
Bank Sta=191.35,237.55
XS Rating Curve= 0 ,0
Exp/Cntr(USF)=0,0
Exp/Cntr=0.3,0.1

Type RM Length L Ch R = 1 ,26106   ,311.4,300,285.1
XS GIS Cut Line= 6
1671032.15517884 459456.060716421671051.94155659459541.294141755
1671068.90116835459614.3514103441671091.51398401459711.760992423
1671108.47326767459784.8185890911671128.25964542459870.052014425
#Sta/Elev= 30
       0  995.38    20.4  981.94    33.8  970.86    47.3  962.82    60.8  950.64
    70.9  940.52    74.2  933.42      81   916.6    84.3  912.79    93.3  905.39
   104.6  892.87   107.9  891.04   111.3  890.79   121.4  892.54   161.8  889.97
   171.9  886.65   185.4  877.08  193.22873.6845   199.9  872.69   239.3  872.99
  242.67873.6837   262.5  878.41   330.2  880.84   340.3  881.96   353.8  885.37
   363.9  892.41   367.3  893.44   407.7  894.41   414.4  897.79     425  906.62
#Mann= 5 ,-1,0
       0      .1       0   127.5     .06       0  193.22    .045       0
  242.67     .06       0   367.5      .1       0
Bank Sta=193.22,242.67
XS Rating Curve= 0 ,0
Exp/Cntr(USF)=0,0
Exp/Cntr=0.3,0.1

Type RM Length L Ch R = 1 ,25806   ,304.2,300,295.3
XS GIS Cut Line= 6
1670649.05555134459644.7726093381670716.48684692459700.533324584
1670774.28528775459748.3281764981670851.34976618459812.054427013
1670909.14820701459859.8489508331670968.88890117 459925.70183751
#Sta/Elev= 30
       0 1006.18    12.2 1003.68    29.2  997.64      42  987.24    56.8  972.43
    68.5  965.32    87.1  946.88    95.4  940.41    98.8  936.21   110.4  918.65
   127.1  899.12   131.4  895.35   167.4  891.38     171  889.27   182.6  878.53
  194.09872.5068     199   871.5   222.3  871.31  231.76872.5069   249.8   876.4
   324.8  880.75   336.4  883.82   355.1  886.08   366.6  893.93   371.3  895.72
   387.5  896.13   396.8  894.85   412.7  894.93   420.1  896.51   426.4  899.65
#Mann= 5 ,-1,0
       0      .1       0   127.5     .06       0  194.09    .045       0
  231.76     .06       0   387.5      .1       0
Bank Sta=194.09,231.76
XS Rating Curve= 0 ,0
Exp/Cntr(USF)=0,0
Exp/Cntr=0.3,0.1

Type RM Length L Ch R = 1 ,25506   ,298.8,300,301.5
XS GIS Cut Line= 6
1670480.02373718459948.8382741661670558.52620484459987.485506594
1670625.81412801460020.6117526741670715.53146826460064.779971421
1670782.81906334460097.9058894221670861.32185909460136.553121835
#Sta/Elev= 30
       0  963.38     6.3  959.44    12.4  954.59    23.3  942.52      36  932.36
      52  917.24    74.5  902.47    85.5  897.33   100.1  889.43   103.5  889.12
   111.1  890.94     133  890.65   142.7  889.78   169.6  879.19   180.6  872.96
  187.77871.2811     199  870.48   221.1  870.25   231.8  870.38  239.97871.2821
   250.1  874.68   257.4  878.83   264.7   881.6     275  887.35     283  888.77
   293.9  894.95   326.5  897.01   356.1   904.9     389  912.11     425  917.85
#Mann= 5 ,-1,0
       0      .1       0      50     .06       0  187.77    .045       0
  239.97     .06       0   322.5      .1       0
Bank Sta=187.77,239.97
XS Rating Curve= 0 ,0
Exp/Cntr(USF)=0,0
Exp/Cntr=0.3,0.1

Type RM Length L Ch R = 1 ,25206   ,640.6,671.7,694.2
XS GIS Cut Line= 6
1670342.76056026460203.0808759181670419.15542059460245.742864087
1670484.63691692460282.3103762571670571.94546933460331.067496583
1670637.42696567460367.6350087521670713.82182601460410.296996921
#Sta/Elev= 30
       0  955.09    13.4  943.25    23.4  936.86    27.1  931.84    34.6  918.83
    42.2  914.11      52  911.42    57.2  908.49    60.9  905.38    69.6  894.48
    76.1  889.65    83.5  887.05   109.9  887.94   150.4   886.1   154.9  884.17
   170.1  873.23  178.23869.9351   207.5  869.08   242.8869.9343   256.3  877.04
   276.2  877.23   290.2  879.25   297.7  883.15   312.4  893.87   316.5  895.26
     339     896     354  900.76   375.1  902.71   392.6  910.78     425  917.11
#Mann= 5 ,-1,0
       0      .1       0      40     .06       0   172.5      .1       0
  178.23    .045       0   242.8      .1       0
Bank Sta=178.23,242.8
XS Rating Curve= 0 ,0
Exp/Cntr(USF)=0,0
Exp/Cntr=0.3,0.1

Type RM Length L Ch R = 1 ,24534   ,216.4,226.7,232.7
XS GIS Cut Line= 2
1670027.01555101460577.6457220851670122.09642688 461038.98316448
#Sta/Elev= 30
       0  917.53    30.7  913.36    40.8  910.47    44.1  907.62    47.5  901.63
    50.8  893.59    54.2  886.84    57.5  883.92    87.7  884.61      91  883.27
   101.1  876.51   107.8  874.22     148  874.84  171.43868.5633   178.1  867.48
   194.9  867.25   228.4  867.68  232.27868.5641   245.1  873.28   258.5   882.8
   271.9  890.04   301.7  897.38   332.3  901.32   348.9   906.9   396.2  916.36
   412.6     923   432.7  935.82   437.6  937.96   452.8  943.17     471  946.37
#Mann= 5 ,-1,0
       0      .1       0      80     .06       0  171.43    .045       0
  232.27     .06       0     270      .1       0
Bank Sta=171.43,232.27
XS Rating Curve= 0 ,0
Exp/Cntr(USF)=0,0
Exp/Cntr=0.3,0.1

Type RM Length L Ch R = 1 ,24308   ,248.8,301.7,327
XS GIS Cut Line= 6
1669874.19522442460581.4462609291669855.99414533460668.946085915
1669844.61359067460743.9462639991669841.30027708460843.946392089
1669841.30027708460918.9462420941669841.30027708461006.446067095
#Sta/Elev= 30
       0  895.01     6.8  892.27    16.8  886.67    26.9  884.66    49.9  884.09
    97.2  887.16   103.8  884.93   111.7  879.62   117.1  876.77   140.3  870.58
  147.93867.8893   156.9  866.98     180  868.23     203  867.39  236.48867.8914
   239.1  868.86   242.9   871.5   252.2  879.54   255.5  881.53   281.7  893.69
     285  896.11   291.6  902.64   301.4  908.96     308  912.08   330.9  919.16
   340.8  925.92     364  938.31   379.9  948.78   406.4   964.4   427.8  975.06
#Mann= 3 ,-1,0
       0     .06       0  147.93    .045       0  236.48      .1       0
Bank Sta=147.93,236.48
XS Rating Curve= 0 ,0
Exp/Cntr(USF)=0,0
Exp/Cntr=0.3,0.1

Type RM Length L Ch R = 1 ,24006   ,164,177,190.9
XS GIS Cut Line= 6
1669807.56838918460524.7777390931669728.98127601460563.253055841
1669661.62117451460596.2316644191669571.80737776460640.202705085
1669504.44694817460673.1813136791669425.85983501460711.656302333
#Sta/Elev= 30
       0  889.74    58.7  886.91   126.6  888.29   137.2  885.85   154.4  874.35
   166.8  868.66   174.1     867  185.55866.7333   199.6  865.58   236.2  865.81
  242.51 866.733     250  869.31   252.5  871.57   254.9  875.23   261.7  891.83
   264.7  896.14   269.6  900.83     280  909.26   301.9  921.86   312.9  935.93
   327.5  947.07   342.1  960.73   350.5  967.37   367.7  977.43   377.5  990.02
   382.4  994.58   389.6  998.22   404.2 1003.06   418.8 1005.24     425 1009.19
#Mann= 5 ,-1,0
       0     .06       0   157.5      .1       0  185.55    .045       0
  242.51     .06       0   312.5      .1       0
Bank Sta=185.55,242.51
XS Rating Curve= 0 ,0
Exp/Cntr(USF)=0,0
Exp/Cntr=0.3,0.1

Type RM Length L Ch R = 1 ,23829   ,123.9,127.2,124.9
XS GIS Cut Line= 6
1669805.36953849460455.1176811741669717.86971349460455.117681174
1669642.86986348460455.1176811741669542.86973541460446.715138925
1669468.14055415460424.2745670061669381.16205357460398.101719094
#Sta/Elev= 30
       0  891.09    22.9  890.32      59  887.28    98.4  887.17   124.6  885.07
   137.7  883.04   170.6  873.64   190.3  867.19  212.74865.3909     243  864.71
   258.7865.4113   266.2  867.64   269.6  870.13   278.4   878.5   288.9  889.71
   296.8  896.65   300.4  896.89   303.9  895.98   307.5  896.72   317.6  907.68
   324.4  913.19   330.3  919.93   331.3  921.32   338.1  935.41   341.5   938.7
   364.5  950.74   372.4  957.24   392.9  970.52   406.6  977.91   431.7  988.89
#Mann= 5 ,-1,0
       0      .1       0    97.5     .07       0  212.74    .045       0
   258.7     .06       0  430.88      .1       0
Bank Sta=212.74,258.7
XS Rating Curve= 0 ,0
Exp/Cntr(USF)=0,0
Exp/Cntr=0.3,0.1

Type RM Length L Ch R = 1 ,23702   ,149.8,144.3,141.3
XS GIS Cut Line= 6
1669817.03785843460338.3224033421669729.53803343460338.322403342
1669654.53818342460338.3224033421669554.53805535460329.919861093
1669479.80887409460307.4792891741669392.83037351460281.306441262
#Sta/Elev= 30
       0  901.17     8.3  897.66    18.2  894.89      28   890.2    34.6  888.86
      51  888.83    80.5  886.22   106.8  883.15     133  878.68   162.5  878.39
   169.1  876.45     179  868.58  191.25864.9827   221.8  864.33   233.2864.9818
   247.2  868.78   264.7  877.25   278.4  885.12   285.2  887.44   305.8  890.03
   329.7  889.78   333.2  890.28   336.6  891.97     340  896.11   346.9  907.75
   360.6  921.61   370.4  937.39   374.3  941.13   405.1  959.34   431.7  971.67
#Mann= 3 ,-1,0
       0      .1       0  191.25    .045       0   233.2     .06       0
Bank Sta=191.25,233.2
XS Rating Curve= 0 ,0
Exp/Cntr(USF)=0,0
Exp/Cntr=0.3,0.1

Type RM Length L Ch R = 1 ,23557   ,195.7,197.8,200
XS GIS Cut Line= 6
1669829.11277458460179.5020809711669741.70940608460183.608371967
  1669666.791905460187.1280499781669566.90201291460191.820953974
1669491.98483992 460195.340631971669404.58114333460199.446922967
#Sta/Elev= 30
       0  911.51    56.6  900.55    89.4  891.57   102.5   886.8   112.4  878.91
   115.7  877.48   145.2  876.28   161.7   876.7   168.2  875.56   171.5  873.27
   178.1  865.85     181864.4879   191.2  863.12   217.5     863  246.26864.4862
   250.3   865.3   256.5  868.76   265.9  878.37   279.9  889.06   309.8  893.52
     339  894.89   352.2  894.59   355.4  896.06   358.7  898.62   375.1  915.46
   385.1  923.82   398.1  936.89   403.9   940.5   414.6     945     425  953.04
#Mann= 4 ,-1,0
       0      .1       0     181    .045       0  246.26      .1       0
   272.5     .06       0
Bank Sta=181,246.26
XS Rating Curve= 0 ,0
Exp/Cntr(USF)=0,0
Exp/Cntr=0.3,0.1

Type RM Length L Ch R = 1 ,23360   ,312.5,316.7,318.9
XS GIS Cut Line= 2
1669830.32395749459993.2252833291669392.39563425459991.337661246
#Sta/Elev= 30
       0  921.01    28.2  917.73      84  903.47    90.5  901.15    97.1  897.39
   116.8  895.04     120  893.42     143  877.39   152.9  874.63   172.5  873.89
   175.8  872.73   182.4  867.18  186.83864.3645   195.5  862.94     248  862.98
  265.11864.3652   284.1  867.87   297.2  868.63   300.5  870.21   310.3  877.06
   339.9   887.3   350.4  894.43   372.7  907.92   375.9  909.16   405.5     911
   408.8   912.8     419  922.83   428.4  930.27   431.7  932.62   437.9   934.9
#Mann= 4 ,-1,0
       0      .1       0  186.83    .045       0  265.11      .1       0
     300     .06       0
Bank Sta=186.83,265.11
XS Rating Curve= 0 ,0
Exp/Cntr(USF)=0,0
Exp/Cntr=0.3,0.1

Type RM Length L Ch R = 1 ,23043   ,248.8,237.1,228.4
XS GIS Cut Line= 4
1669819.25218701459681.6328685941669688.75230127459691.205750064
 1669464.1252734 459662.891418821669342.22294918459678.602672025
#Sta/Elev= 30
       0  944.91    20.4   937.1    33.6  929.29      50   916.8    66.5  914.51
    86.2  901.03   106.2  896.85   125.7  895.21   139.9  900.29   152.1  900.26
   162.1  893.28   181.9  874.46   195.1  870.94  207.76864.2041   218.3  862.72
   261.3  862.69  271.07864.2034   284.4  865.92   297.6   865.3   304.2  867.91
   314.2     875   324.1  877.73   390.2     874   393.5  875.83   401.1  884.91
   406.8  889.36   416.7  902.87   429.9  914.58   446.5  923.18   480.2  936.93
#Mann= 4 ,-1,0
       0      .1       0  207.76    .045       0  271.07      .1       0
  477.26     .07       0
Bank Sta=207.76,271.07
XS Rating Curve= 0 ,0
Exp/Cntr(USF)=0,0
Exp/Cntr=0.3,0.1

Type RM Length L Ch R = 1 ,22806   ,279.5,271.1,263.9
XS GIS Cut Line= 6
1669748.05899376459400.6910765021669662.30325976 459418.07391575
1669588.79815742 459432.973492251669490.79146367 459452.83959426
1669417.28603326 459467.739170761669331.53029926459485.122010008
#Sta/Elev= 30
       0  943.71    11.8  937.02    18.5  932.21    31.9  918.88    35.2  916.34
    45.2  910.14    55.3   905.5    58.6  902.91      62  898.78    65.3  892.89
      72  879.07    75.4  875.43    85.4  869.89    88.8  868.57    95.5  867.69
   152.4  868.13   162.4  869.08  175.37863.9606   182.5  863.15   252.8  863.07
  254.89863.9633   266.2  866.37     293  865.78   319.7  869.21   329.6  876.57
   339.8   881.3   357.5  891.78   396.7  912.78   406.8  915.92     425  918.07
#Mann= 3 ,-1,0
       0      .1       0  175.37    .045       0  254.89      .1       0
Bank Sta=175.37,254.89
XS Rating Curve= 0 ,0
Exp/Cntr(USF)=0,0
Exp/Cntr=0.3,0.1

Type RM Length L Ch R = 1 ,22535   ,472.1,392.2,349.7
XS GIS Cut Line= 2
1669681.25612134459106.1627019151669272.96855208459254.082681666
#Sta/Elev= 30
       0  956.91     7.5  956.08    27.8  948.92    40.6  943.59    48.3  938.73
    56.4  931.12    70.3  913.79    80.8  904.28    91.3  893.02    94.7  888.46
   101.7  877.42   104.6  874.15   112.3  868.38   119.2  866.24   147.1  866.59
   150.6   865.9   155.9  863.52     161  862.47   171.2  862.25   222.5  863.38
   262.2  860.94   269.2  861.61   273.2  863.52   276.2  865.63   283.9  867.53
   332.6  869.86   377.4  883.32   391.9   890.4   406.9  892.68   434.3  906.54
#Mann= 3 ,-1,0
       0      .1       0   155.9    .045       0   273.2      .1       0
Bank Sta=155.9,273.2
XS Rating Curve= 0 ,0
Exp/Cntr(USF)=0,0
Exp/Cntr=0.3,0.1

Type RM Length L Ch R = 1 ,22143   ,221.3,213.9,206.9
XS GIS Cut Line= 6
1669126.57946985458830.1330442461669161.04692061458910.558408323
1669190.59082478458979.4946221591669228.73641778459071.942928079
 1669219.7042836459156.3374443231669205.00261401459264.645298573
#Sta/Elev= 30
       0  964.94    10.1  959.37    17.2  952.29    26.8  940.85    36.8  932.28
    39.3  929.45    45.8  918.06    49.3  914.27    60.1  907.97    69.3  899.06
    81.8  888.65    88.6  885.29   101.8  881.93   138.6  874.36   156.4  871.84
   167.1  863.11  175.35859.4543   181.3  858.48   199.4  858.34   220.4  858.52
  225.24 859.452   237.1  867.09   248.8  871.12   279.4  872.16   299.2  875.06
   355.3   880.6   401.7  897.22   421.5  900.11   438.1   907.6   456.7  909.13
#Mann= 3 ,-1,0
       0      .1       0  175.35    .045       0  225.24      .1       0
Bank Sta=175.35,225.24
XS Rating Curve= 0 ,0
Exp/Cntr(USF)=0,0
Exp/Cntr=0.3,0.1
